HEC-RAS study W156-00-00.prj: W156-00-00

--- W156-00-00.g02 (geometry) --- (continued)

Type RM Length L Ch R = 1 ,9776.550,143.92,180.78,207.37
BEGIN DESCRIPTION:
d/s face of Brittmore Dr. Bridge
END DESCRIPTION:
XS GIS Cut Line= 4
     3056827.828    13846076.093      3056383.47    13846599.169
      3056426.99    13846714.186     3055517.766    13847918.054
#Sta/Elev= 30
       0   75.45  37.802   73.57 133.212   77.39 236.534   76.36 282.949   73.24
 319.336   76.49  353.61   76.94  465.51   72.93 509.272   73.71  529.34   68.99
 544.939   61.31 551.233    59.6 557.745   59.85 563.084   61.95 568.918   65.51
 572.276   71.34 585.619   75.24 646.812   75.52 684.614   72.17 712.368   74.04
 958.568   77.071004.021   74.531175.254   75.231215.205   76.961320.451   75.92
1383.235   78.621437.237    79.51465.394   82.57 1535.73   81.751639.038   82.72
#Mann= 3 ,-1 , 0
       0     .99       0 509.272    .035       0 585.619     .99       0
#XS Ineff= 2 , 0
       0 509.272   75.35 585.619       0   75.35
Permanent Ineff=
       F       F
#Block Obstruct= 1 ,-1
       0 122.987   77.18
Bank Sta=509.272,585.619
XS Rating Curve= 0
Skew Angle= 45
Exp/Cntr=.5,.3

Type RM Length L Ch R = 1 ,9586.862,350.79,392.38,407.52
XS GIS Cut Line= 2
     3056928.602    13845592.565     3055300.037    13847968.066
#Sta/Elev= 30
       0   76.09   91.01    73.9  170.97   77.81  197.92   74.82  404.13   75.41
  472.93   74.04  503.22   75.89  717.71   75.23  778.32   76.72  841.34   72.55
  1022.9   75.84 1130.43   73.84 1160.75   71.21 1186.71   59.12 1202.13   61.53
 1213.71   69.16 1215.44   72.92 1216.94   73.21 1277.98   75.57 1370.03   71.77
  1422.7   74.55 1501.16   75.87 1730.24   76.06 1868.83   74.08 1915.48   75.96
 1988.87   74.53 2175.42   77.51 2232.27   76.37 2366.83   80.93 2880.14   83.38
#Mann= 3 ,-1 , 0
       0     .99       0 1130.43    .035       0 1216.94     .99       0
#Block Obstruct= 1 ,-1
       0  170.97   77.81
Bank Sta=1130.43,1216.94
XS Rating Curve= 0
Exp/Cntr=.3,.1

Type RM Length L Ch R = 1 ,9192.376,413.51,468.57,491.47
XS GIS Cut Line= 4
     3056544.697    13845624.447     3056011.924    13846280.364
     3055961.904    13846313.511     3055087.316    13847461.276
#Sta/Elev= 30
       0   75.04   36.31   73.73    92.7   76.08  219.59   76.15  287.49   77.05
  525.26   73.29  595.21   74.27  758.06   72.92  844.71    73.2  873.49   70.75
  879.49   67.85  880.49   64.92  888.88   60.75  889.91   58.82  899.27   57.99
   901.7    58.2  904.49   62.25  930.98      72  950.59    73.3 1085.67   72.22
 1246.78    76.4 1269.08    75.7 1299.96   76.83 1432.47   74.78 1478.26   79.15
 1508.34   75.33 1642.87   74.31 1956.14   76.09 2068.57   81.04 2348.04   81.05
#Mann= 3 ,-1 , 0
       0     .99       0  844.71    .035       0  950.59     .99       0
#Block Obstruct= 1 ,-1
       0    92.7   76.08
Bank Sta=844.71,950.59
XS Rating Curve= 0
Exp/Cntr=.3,.1

Type RM Length L Ch R = 1 ,8724.199,64.36,80.36,85.44
BEGIN DESCRIPTION:
I
END DESCRIPTION:
XS GIS Cut Line= 4
     3056447.313    13845468.196      3055627.84    13845985.839
     3055600.079    13846036.978      3054902.71    13846749.338
#Sta/Elev= 30
       0   75.89  102.59   75.67  152.82   76.82  208.58   76.73  345.35   74.11
  366.19   74.37  430.59   76.75  564.83   75.22  618.97   75.52  672.19   71.85
   804.7   73.13  905.64   72.01  924.29   73.39  974.62   74.64  974.83   74.65
  982.69   71.34  998.01   66.75 1005.01   63.75 1010.01   58.89 1013.99   58.46
 1020.96   58.88 1032.01   64.85 1049.72   71.43 1121.91   73.73 1212.96   72.12
 1351.48   73.25 1371.23   72.69 1865.63      75 1909.25   76.82 2024.35   76.44
#Mann= 3 ,-1 , 0
       0     .99       0  974.83    .035       0 1049.72     .99       0
Bank Sta=974.62,1049.72
XS Rating Curve= 0
Exp/Cntr=.5,.3

Type RM Length L Ch R = 1 ,8635.686,36.39,34.22,34.91
BEGIN DESCRIPTION:
u/s face of Rummel Cr. Dr. Bridge
END DESCRIPTION:
XS GIS Cut Line= 4
     3056392.771    13845429.739     3055577.139    13845949.879
      3055525.85    13845981.368     3054847.524    13846711.117
#Sta/Elev= 30
       0    75.6  138.47   74.73   234.9    76.9  386.64   73.89  441.57   75.05
  521.17   75.47  555.97   75.24  609.34   72.18  805.18   74.72  977.91   71.43
  982.78   70.15  998.41   68.88 1011.84   61.97 1014.96   60.71 1016.46   60.76
 1018.75   58.99 1022.54   58.02 1028.35   58.63 1030.21   60.76 1034.75   61.71
 1039.93   63.83 1052.49   70.54 1061.97   71.76 1105.77   71.71 1254.54   73.66
 1393.23   74.25 1438.87   72.92 1902.23   75.24 1964.72   77.89 2023.88   76.67
#Mann= 3 ,-1 , 0
       0     .99       0  977.91    .035       0 1061.97     .99       0
#XS Ineff= 2 , 0
       0  980.13   71.48 1054.12       0   71.76
Permanent Ineff=
       F       F
Bank Sta=977.91,1061.97
XS Rating Curve= 0
Exp/Cntr=.5,.3

Type RM Length L Ch R = 3 ,8619.259,,,
BEGIN DESCRIPTION:
Rummel Cr. Dr. Bridge
END DESCRIPTION:
Bridge Culvert--1,0,-1,-1, 0
Deck Dist Width WeirC Skew NumUp NumDn MinLoCord MaxHiCord MaxSubmerge Is_Ogee
.01,34.2,2.6,0, 2, 2, 72.55, , .95, 0, 0,0,,
     977    1062
   72.55   72.55
   70.75   70.75
     977    1062
   72.55   72.55
   70.75   70.75
BR Coef=-1 , 0 , 0 ,, 0 ,,,.8,-1,,0,
WSPro=,,,, 1 ,,,, 0 ,,,, 0 ,,,,-1 ,-1 ,-1 , 0 , 0 , 0 , 0 , 0
BC Design=,, 0 ,, 0 ,,,,,,
BC HTab HWMax=77.91

Type RM Length L Ch R = 1 ,8601.774,73.25,72.13,69.11
BEGIN DESCRIPTION:
d/s face of Rummel Cr. Dr. Bridge
END DESCRIPTION:
XS GIS Cut Line= 4
     3056365.464    13845407.899     3055549.832    13845928.038
     3055498.543    13845959.528     3054820.217    13846689.276
#Sta/Elev= 30
       0   75.62  158.79   74.37  264.69   76.52  427.26   73.59   508.8   74.42
  551.93   73.73  576.96   72.36  754.81   74.99  967.37   72.69  974.94   72.44
  990.24   68.88 1003.67   61.97 1006.79   60.71 1008.29   60.76 1010.58   58.99
 1014.37   58.02 1020.18   58.63 1022.04   60.76 1026.58   61.71 1031.76   63.83
 1044.32   70.54 1054.86   72.28 1061.26   72.56 1135.56   73.83 1194.64   73.27
 1412.09   74.67 1468.69   73.02 1922.67   75.36 1939.44   76.07 2023.87   76.47
#Mann= 3 ,-1 , 0
       0     .99       0  967.37    .035       0 1061.26     .99       0
#XS Ineff= 2 , 0
       0  981.51   72.55 1045.59       0   72.55
Permanent Ineff=
       F       F
#Block Obstruct= 2 , 0
       0     610    72.9               0
Bank Sta=967.37,1061.26
XS Rating Curve= 0
Exp/Cntr=.5,.3

Type RM Length L Ch R = 1 ,8533.452,118.18,148.42,154.48
XS GIS Cut Line= 4
     3056378.382    13845379.025      3055492.56     13845870.99
     3055454.124    13845911.233     3054778.008    13846617.835
#Sta/Elev= 30
       0   75.85  217.56   74.15  318.21   75.94  357.17   76.27  431.81   75.36
  485.43   74.18  508.12   73.16  571.22   72.53  659.64   74.82   711.3   75.49
  814.31      74 1017.64   73.42 1022.45   73.25  1058.5   66.15 1068.26   60.19
 1069.74   58.99 1073.53   58.02 1079.34   58.63  1080.5   59.55 1089.97   61.23
 1094.74   73.05 1096.81   73.18 1264.83   73.58 1327.79   74.29 1502.73   75.53
 1582.95   73.22 1877.14   74.66 1946.07   75.98 2004.92   75.85 2046.88   76.28
#Mann= 3 ,-1 , 0
       0     .99       0 1017.64    .035       0 1096.81     .99       0
#Block Obstruct= 2 , 0
       0     575   72.65               0
Bank Sta=1017.64,1096.81
XS Rating Curve= 0
Exp/Cntr=.3,.1

Type RM Length L Ch R = 1 ,8386.468,32.09,30.54,29.93
BEGIN DESCRIPTION:
H
H
END DESCRIPTION:
XS GIS Cut Line= 4
     3055880.712    13845602.335     3055377.745    13845774.417
     3055339.677    13845819.936     3054936.008    13846211.634
#Sta/Elev= 30
       0   72.65   17.66    72.7   50.83   73.75  121.88   74.08  125.77   73.47
  201.72   74.44  273.87   73.32  323.93   73.22  389.75   75.64  540.86   72.95
  565.26   65.35  575.26   64.45   575.8    59.1  577.26   57.82  580.24   57.18
  589.12   57.07  595.21   57.56  605.44   62.33  617.49   71.07  634.78    72.6
  705.71    71.3  730.47   71.33  758.25   71.69  871.94   74.39   953.8   74.29
  958.66   73.79  977.49   74.71  996.88   74.03 1069.24   73.07  1153.4   73.36
#Mann= 3 ,-1 , 0
       0     .99       0  540.86    .035       0  634.78     .99       0
Bank Sta=540.86,634.78
XS Rating Curve= 0
Exp/Cntr=.5,.3

Type RM Length L Ch R = 1 ,8356.165,3.76,4.05,3.97
BEGIN DESCRIPTION:
u/s of 42" steel pipeline # 2
END DESCRIPTION:
XS GIS Cut Line= 4
     3055856.795    13845584.013     3055353.912    13845755.834
     3055315.845    13845801.354     3054912.175    13846193.051
#Sta/Elev= 27
       0   72.61     6.3   72.85  104.21   72.89  281.63    73.2  359.84   76.07
  487.47   73.83  546.82   72.69   558.4   67.59  572.88   64.45  576.88   59.75
  578.88   57.75  585.88   57.25  592.88   57.65  594.88   58.85  607.11   63.05
   621.2   69.28  628.33   72.91  635.35    72.5  638.94   72.87  698.59   71.75
  713.17   70.74  743.38   72.04  858.13   74.76   930.3   74.67  950.32   74.99
 1018.69   72.96 1153.24   73.54
#Mann= 3 ,-1 , 0
       0     .99       0  546.82    .035       0  628.33     .99       0
Bank Sta=546.82,628.33
XS Rating Curve= 0
Exp/Cntr=.5,.3

Type RM Length L Ch R = 3 ,8354.151,,,
BEGIN DESCRIPTION:
42" steel pipeline # 2
END DESCRIPTION:
Bridge Culvert--1,0,-1,-1, 0
Deck Dist Width WeirC Skew NumUp NumDn MinLoCord MaxHiCord MaxSubmerge Is_Ogee
.01,3.5,3,0, 2, 2, 70.95, , .95, 0, 0,0,,
  546.88  626.88
   70.95   70.95
   67.45   67.45
  548.58  628.58
   70.95   70.95
   67.45   67.45
BR Coef=-1 , 0 , 0 ,, 0 ,,,.8,0,,0,
WSPro=,,,, 1 ,,,, 0 ,,,, 0 ,,,,-1 ,-1 ,-1 , 0 , 0 , 0 , 0 , 0
BC Design=,, 0 ,, 0 ,,,,,,
BC HTab HWMax=76.07

Type RM Length L Ch R = 1 ,8352.148,64.35,140.88,297.15
BEGIN DESCRIPTION:
d/s of 42" steel pipeline # 2
END DESCRIPTION:
XS GIS Cut Line= 4
      3055856.05    13845581.845     3055350.758    13845753.366
      3055312.69    13845798.886     3054909.021    13846190.584
#Sta/Elev= 28
       0   72.57    8.57   72.89  103.79   72.94  278.74    73.2  358.27   76.12
  485.36   73.89  549.83   72.65  559.28   68.49  575.31   60.61  578.58   59.75
  580.58   57.75  587.58   57.25  594.58   57.65  596.58   58.85  599.58   59.85
  608.81   62.68  618.98   67.18  630.03    72.8  636.25   72.43  640.64   72.89
   695.1   71.87  712.69   70.65  749.11   72.21  858.52   74.81  927.32   74.73
  946.41   75.03 1017.08   72.95 1155.42   73.56
#Mann= 3 ,-1 , 0
       0     .99       0  549.83    .035       0  630.03     .99       0
Bank Sta=549.83,630.03
XS Rating Curve= 0
Exp/Cntr=.5,.3

Type RM Length L Ch R = 1 ,8205.582,241,277.56,427.28
XS GIS Cut Line= 5
     3055661.439     13845633.34     3055293.501    13845676.979
     3055260.893    13845677.273     3055220.449    13845677.637
     3054693.143     13845741.45
#Sta/Elev= 27
       0   73.42   20.73   73.55   47.69   73.58  100.25   72.92  162.42   75.23
  247.69   74.91  250.38   74.79  258.27   74.87  370.01   73.02   402.1   63.45
   412.1   62.55   416.1   57.85   418.1   55.85   425.1   55.35   432.1   55.75
   434.1   56.95   437.1   57.95   443.5    65.5  460.13   72.86  474.61   72.83
  498.93   72.63  785.63   73.17  793.49   73.22  849.36   74.17  862.36    73.8
  935.65   73.27  974.72   73.61
#Mann= 3 ,-1 , 0
       0     .99       0  370.01    .035       0  460.13     .99       0
Bank Sta=370.01,460.13
XS Rating Curve= 0
Exp/Cntr=.3,.1

Type RM Length L Ch R = 1 ,7924.317,61.54,95.57,174.51
BEGIN DESCRIPTION:
G
END DESCRIPTION:
XS GIS Cut Line= 4
     3055672.073     13845618.69      3055334.66     13845416.42
     3055245.459    13845390.396     3054438.927    13845012.148
#Sta/Elev= 30
       0   73.65   35.98    74.1  144.71   73.25  196.55   74.58  283.23   73.44
  302.05   74.98  360.19   73.79  370.84   74.36  393.86   73.11  417.14   70.68
  425.56   66.44  430.49   61.75  435.06   56.42  438.23   55.59  451.37   54.85
     456   56.86  458.49   60.45  462.49   64.25   479.8   69.05  489.49   70.21
  576.55   72.93  649.86   73.51  801.58   71.95  843.65   72.96  987.36   75.14
 1130.81   71.79 1180.32    71.1  1189.8   71.77 1308.82   76.46 1377.14   75.65
#Mann= 3 ,-1 , 0
       0     .99       0  393.86    .035       0  576.55     .99       0
Bank Sta=393.86,576.55
XS Rating Curve= 0
Exp/Cntr=.5,.3

Type RM Length L Ch R = 1 ,7827.230,4.33,4.05,4.21
BEGIN DESCRIPTION:
u/s of 42" pipeline #1
END DESCRIPTION:
XS GIS Cut Line= 4
     3055628.036    13845566.044      3055375.04    13845348.042
     3055298.264    13845294.223     3054556.878    13844708.236
#Sta/Elev= 30
       0   74.11   45.63   73.84   74.16    74.8  211.39   73.37  291.62   71.54
  302.33   71.04  343.37   70.84  347.62   70.26   352.1   67.96  375.75   61.75
  379.75   56.85  385.75   56.55  391.75   56.95  392.75   58.45  403.75   60.45
  407.75   64.25  421.15   71.92  497.68   73.41  599.62   72.45  777.31   72.32
  938.28   75.15  964.81   76.03  1058.6   72.32  1064.1   72.26 1080.06   72.36
 1092.36   72.88 1195.49   75.45 1246.33   74.28  1315.3   72.07 1372.73    73.2
#Mann= 3 ,-1 , 0
       0     .99       0  343.37    .035       0  421.15     .99       0
Bank Sta=343.37,421.15
XS Rating Curve= 0
Exp/Cntr=.5,.3

Type RM Length L Ch R = 3 ,7825.141,,,
BEGIN DESCRIPTION:
42" steel pipeline # 1
END DESCRIPTION:
Bridge Culvert--1,0,-1,-1, 0
Deck Dist Width WeirC Skew NumUp NumDn MinLoCord MaxHiCord MaxSubmerge Is_Ogee
.02,3.5,3,0, 2, 2, 69.35, , .95, 0, 0,0,,
  346.75  429.75
   69.35   69.35
   65.85   65.85
  344.65  427.65
   69.35   69.35
   65.85   65.85
BR Coef=-1 , 0 , 0 ,, 0 ,,,.8,0,,0,
WSPro=,,,, 1 ,,,, 0 ,,,, 0 ,,,,-1 ,-1 ,-1 , 0 , 0 , 0 , 0 , 0
BC Design=,, 0 ,, 0 ,,,,,,
BC HTab HWMax=76.03

Type RM Length L Ch R = 1 ,7823.121,47.69,91.94,136.75
BEGIN DESCRIPTION:
d/s of 42" pipeline #1
END DESCRIPTION:
XS GIS Cut Line= 4
      3055630.42    13845562.784     3055377.424    13845344.782
     3055300.648    13845290.962     3054559.262    13844704.976
#Sta/Elev= 30
       0   74.15   42.02   73.91   69.17   74.82  213.02   73.32  290.69   71.55
  304.32    70.9  310.41   70.97  344.66   70.64  345.51   70.52  371.94   59.95
  377.65   56.85  383.65   56.55  389.65   56.95  390.65   58.45  401.65   60.45
  405.65   64.25  420.52   71.94   495.9   73.39  594.36   72.47  780.35   72.33
  933.02   75.03  962.76   76.02 1052.26   72.48 1067.14   72.32 1076.24   72.38
 1083.26   72.68 1196.43   75.49 1244.29   74.39 1316.61   72.07 1372.73   73.18
#Mann= 3 ,-1 , 0
       0     .99       0  344.66    .035       0  420.52     .99       0
Bank Sta=344.66,420.52
XS Rating Curve= 0
Exp/Cntr=.5,.3

Type RM Length L Ch R = 1 ,7730.294,308.17,291.07,285.28
XS GIS Cut Line= 4
     3055705.185     13845625.56      3055430.94    13845294.544
     3055384.149    13845211.658     3054661.989     13844530.76
#Sta/Elev= 30
       0   73.21   69.44   74.47  123.51   74.26  140.16   74.94  343.83   72.61
  383.76    71.7  425.62   69.63  441.07   65.18  449.12   63.57  454.48   61.75
  459.75   56.07  472.74   55.54  474.79   55.91  476.59   57.37  482.48   60.45
  486.48   64.25  494.82    65.4   511.8   72.34  565.25   72.97  926.01   73.17
 1020.03   72.81 1072.59   74.67  1132.2   75.38 1218.21   74.14 1272.44   75.48
 1362.01   72.87  1381.4   72.82 1413.21   72.24 1475.93   72.97 1517.59   73.01
#Mann= 3 ,-1 , 0
       0     .99       0  343.83    .035       0   511.8     .99       0
Bank Sta=343.83,511.8
XS Rating Curve= 0
Exp/Cntr=.3,.1

Type RM Length L Ch R = 1 ,7440.611,39.11,35.13,26.6
BEGIN DESCRIPTION:
F
END DESCRIPTION:
XS GIS Cut Line= 4
     3056049.293    13845518.493     3055685.493    13845155.954
     3055644.576     13845090.18     3054926.983    13844360.716
#Sta/Elev= 30
       0   75.39   75.55   73.91  415.46   71.22  435.66    71.3  478.88   70.01
  500.28   67.94  516.58   63.65  528.78   62.85  535.78   58.01  537.66   53.98
  539.71   53.75  550.24   53.91  552.64   54.16  554.76      58  555.78   60.35
  566.78   63.15  583.79   70.85   597.6    72.2  613.44   72.29   706.9   72.86
  848.33   74.13  893.74   74.78  952.97   74.42  1087.6   74.21 1292.84   74.54
 1420.85   74.05 1440.31   73.67 1495.51   73.58 1545.37   74.77 1614.32   75.19
#Mann= 3 ,-1 , 0
       0     .99       0  435.66    .035       0  613.44     .99       0
Bank Sta=435.66,597.6
XS Rating Curve= 0
Exp/Cntr=.5,.3

Type RM Length L Ch R = 1 ,7404.722,2.04,2,2.02
BEGIN DESCRIPTION:
u/s side of 14" steel pipeline
END DESCRIPTION:
XS GIS Cut Line= 2
     3056082.094    13845506.561     3054953.947    13844343.413
#Sta/Elev= 30
       0   75.12   59.93   73.83  164.48   73.71  424.02   71.48  442.51   71.69
  506.99   67.24   516.9   64.59  530.38   63.63  534.06   62.02  537.21   59.87
     540    57.2  541.14   56.65  543.05   53.93  545.12   53.74  550.05   54.05
  551.42   55.34   551.6   56.02  567.35   59.01  572.75   63.43  583.18   65.05
  591.65   70.65  608.79   72.46  615.74   72.51  922.51   74.96    1063   74.45
 1303.83   74.84 1429.44    74.3 1461.16   73.68 1552.12   73.54 1620.38   74.42
#Mann= 3 ,-1 , 0
       0     .99       0  442.51    .035       0  615.74     .99       0
Bank Sta=442.51,608.79
XS Rating Curve= 0
Exp/Cntr=.5,.3

Type RM Length L Ch R = 3 ,7403.695,,,
BEGIN DESCRIPTION:
14" steel pipeline
END DESCRIPTION:
Bridge Culvert--1,0,-1,-1, 0
Deck Dist Width WeirC Skew NumUp NumDn MinLoCord MaxHiCord MaxSubmerge Is_Ogee
.01,1.94,3,0, 2, 2, 59.98, , .95, 0, 0,0,,
   439.8   639.8
   59.98   59.98
   58.48   58.48
  439.69  639.69
   59.98   59.98
   58.48   58.48
BR Coef=-1 , 0 , 0 ,, 0 ,,,.8,0,,0,
WSPro=,,,, 1 ,,,, 0 ,,,, 0 ,,,,-1 ,-1 ,-1 , 0 , 0 , 0 , 0 , 0
BC Design=,, 0 ,, 0 ,,,,,,
BC HTab HWMax=75.12

Type RM Length L Ch R = 1 ,7402.695,68.87,67.39,68.17
BEGIN DESCRIPTION:
d/s side of 14" steel pipeline
END DESCRIPTION:
XS GIS Cut Line= 2
     3056083.677    13845505.377      3054955.63    13844342.333
#Sta/Elev= 30
       0   75.08   57.65   73.84  170.21   73.71  424.48   71.52  444.79   71.76
  505.34   67.57  516.85   64.53  530.27   63.63  533.95   62.02   537.1   59.87
  539.89    57.2  541.03   56.65  542.94   53.93  545.01   53.74  549.94   54.05
  551.31   55.34  551.49   56.02  567.24   59.01  572.64   63.43  583.07   65.05
  591.55   70.63  608.94   72.49  791.18    73.6  923.97   74.97 1060.63   74.46
 1305.53   74.85 1429.44   74.32 1461.96   73.68 1555.21   73.54 1620.24   74.37
#Mann= 3 ,-1 , 0
       0     .99       0  444.79    .035       0  608.94     .99       0
Bank Sta=444.79,608.94
XS Rating Curve= 0
Exp/Cntr=.5,.3

Type RM Length L Ch R = 1 ,7335.563,628.48,579.46,590.93
XS GIS Cut Line= 2
     3056142.805    13845471.423     3055012.374    13844305.921
#Sta/Elev= 30
       0   74.08  121.32   74.25  174.52   73.09  371.76   73.64   448.3   72.98
  469.68   73.22  478.93   73.59  496.26   73.16  511.57   70.55  545.36    60.1
  548.86   58.21  551.72   54.02  556.97   53.72   563.8   54.25  566.01   54.49
  568.54   58.31  568.86   60.35  579.86   63.15  599.41   70.78  607.59    71.5
  622.34   73.22  981.29    75.4 1001.35   75.08 1076.03   74.64 1320.74   74.65
 1329.47   73.79 1371.06   75.16 1437.82   74.87 1497.23    73.7 1623.66    73.5
#Mann= 3 ,-1 , 0
       0      .1       0  496.26    .035       0  622.34     .99       0
Bank Sta=496.26,622.34
XS Rating Curve= 0
Exp/Cntr=.3,.1

Type RM Length L Ch R = 1 ,6756.135,300.87,250.63,141.44
XS GIS Cut Line= 4
     3057522.664    13845587.549     3056214.146    13844718.265
      3056162.78    13844653.614     3055864.586    13844381.356
#Sta/Elev= 30
       0   77.47  131.62   76.24  244.66   76.97  370.32   73.65  428.53   74.37
  527.11   77.41  545.39   77.56  776.29   76.32  805.13   74.74  912.47   73.27
 1042.26   74.35 1077.18   73.11 1253.43   73.52 1487.08   72.45 1499.49   72.29
 1521.97   69.05 1553.33   65.91 1594.38   59.95 1596.38   57.37  1598.4   53.37
 1603.52    53.1 1613.44   53.36 1615.34   57.39 1621.38   60.35 1653.52   70.13
 1666.42   71.55 1695.55   73.84 1851.64   73.64 1996.09   74.85 2057.31   72.64
#Mann= 3 ,-1 , 0
       0     .99       0 1487.08    .035       0 1666.42     .99       0
Bank Sta=1487.08,1695.55
XS Rating Curve= 0
Exp/Cntr=.3,.1

Type RM Length L Ch R = 1 ,6503.973,165.54,59.44,52.38
BEGIN DESCRIPTION:
E
END DESCRIPTION:
XS GIS Cut Line= 4
     3057587.911    13845118.632     3056290.654    13844472.909
     3056154.571    13844471.571     3055928.793    13844328.632
#Sta/Elev= 30
       0   77.24  216.56   75.13  296.87   78.17  394.07    75.5  417.66   76.22
  606.15   76.21  754.02   72.23  873.77   74.84   917.1   73.87  948.33   74.85
 1085.55   74.03 1140.34   71.53 1155.92   72.32 1264.34   73.11 1325.89   70.92
 1352.25   60.99 1356.59   57.43 1360.64   57.26 1362.53   53.38 1372.73   52.84
 1377.86    53.4 1380.59   57.75  1383.6   60.08 1417.29   69.99 1487.36   72.31
 1593.06   73.14  1649.5   73.47 1758.17   71.75 1809.48   76.08 1852.39   73.81
#Mann= 4 ,-1 , 0
       0     .99       0 1325.89    .035       0 1417.29      .2       0
 1593.06     .99       0
Bank Sta=1325.89,1417.29
XS Rating Curve= 0
Exp/Cntr=.5,.3

Type RM Length L Ch R = 1 ,6446.272,71.46,80.81,67.21
BEGIN DESCRIPTION:
u/s face of Memorial Dr. Br.
END DESCRIPTION:
XS GIS Cut Line= 3
     3056799.197    13844467.412     3056238.184    13844447.357
     3055948.168    13844309.751
#Sta/Elev= 30
       0   72.72  71.623   72.71  86.217   73.47 172.387   72.57  227.81   71.74
 248.521   71.86 281.203   70.29 344.181   69.48  349.03   68.89 357.487   67.25
 372.203   55.21 376.112   53.38 379.664   53.03 385.697   52.84 388.553   53.38
 389.672   55.21 399.426   61.29 412.234    60.7  433.79   65.99  444.54   69.35
 486.169    71.8 506.532   72.33 569.416   72.81 643.962   70.48 650.709   70.44
 689.293   72.84 746.125    74.2 770.501   73.79 781.975   75.04 829.166   75.16
#Mann= 3 ,-1 , 0
       0     .99       0 344.181    .035       0  444.54     .99       0
#XS Ineff= 2 , 0
       0  349.03   72.75 442.623       0   72.75
Permanent Ineff=
       F       F
Bank Sta=344.181,444.54
XS Rating Curve= 0
Skew Angle= 20
Exp/Cntr=.5,.3

Type RM Length L Ch R = 3 ,6403.377,,,
BEGIN DESCRIPTION:
Memorial Dr. Bridge
END DESCRIPTION:
Bridge Culvert--1,0,-1,-1, 0
Deck Dist Width WeirC Skew NumUp NumDn MinLoCord MaxHiCord MaxSubmerge Is_Ogee
.15,71.05,2.6,20, 2, 2, 72.75, , .95, 0, 0,0,,
 248.521 506.532
   72.75   72.75
   68.75   68.75
 262.588 460.976
   72.75   72.75
   68.75   68.75
Pier Skew, UpSta & Num, DnSta & Num=  ,371.32, 4 ,345.967, 4 , 3 , 3 , 0 ,,
    1.12    1.12    2.65    2.65
   51.25   66.11   66.11   68.75
    1.12    1.12    2.65    2.65
   51.25   66.11   66.11   68.75
Pier Skew, UpSta & Num, DnSta & Num=  ,401.409, 4 ,373.34, 4 , 3 , 3 , 0 ,,
    1.12    1.12    2.65    2.65
   51.25   66.11   66.11   68.75
    1.12    1.12    2.65    2.65
   51.25   66.11   66.11   68.75
BR Coef=-1 , 1 , 1 ,1.25, 0 ,,,.8,-1,2,0,
WSPro=,,,, 1 ,,,, 0 ,,,, 0 ,,,,-1 ,-1 ,-1 , 0 , 0 , 0 , 0 , 0
BC Design=,, 0 ,, 0 ,,,,,,
BC HTab HWMax=75.16

Type RM Length L Ch R = 1 ,6367.704,67.9,167.58,235.89
BEGIN DESCRIPTION:
d/s face of Memorial Dr. Br
END DESCRIPTION:
XS GIS Cut Line= 3
     3056811.038    13844398.728     3056250.026    13844378.673
     3055976.118    13844250.173
#Sta/Elev= 30
       0   70.31  58.327   69.72  74.903   70.88 123.269   70.84 142.955   71.16
 149.815    71.9 164.324   68.53 193.868   68.66 227.584   72.63 262.588   72.55
 279.728   70.31  288.58   67.92 323.395   63.61 329.334    63.6 340.413   62.43
 347.094   60.22 354.396   55.21 358.305   53.38  367.89   52.84 370.746   53.38
 371.865   55.21 378.828   56.22 386.777   59.36 410.937   66.05 420.231   66.13
 442.764   71.71 460.976   72.52 620.075    73.2 690.542   74.92 811.819   73.42
#Mann= 5 ,-1 , 0
       0     .99       0 262.588     .07       0 358.305    .035       0
 370.746     .07       0 442.764     .99       0
#XS Ineff= 2 , 0
       0 285.488   72.75 430.821       0   72.75
Permanent Ineff=
       F       F
Bank Sta=262.588,442.764
XS Rating Curve= 0
Skew Angle= 20
Exp/Cntr=.5,.3

Type RM Length L Ch R = 1 ,6195.197,108.29,175.28,234.96
XS GIS Cut Line= 2
     3056838.064    13844409.692     3056231.638    13844117.834
#Sta/Elev= 30
       0   70.69   98.84   69.51  140.74   71.26  171.44   71.13  209.34   68.08
  219.72   66.26  232.01   65.82  256.26   60.09  267.82   59.21   298.6   59.52
   314.5   55.74  328.57   49.89  331.89   49.19  341.76   50.15  344.57   52.15
  360.46   55.92  362.36   55.42  377.52   59.46  394.17   65.02  439.12   70.13
  442.87   70.19  465.58   66.42  476.41   67.76  515.01   68.75  539.14   68.14
   548.3   68.97  573.98   69.27  614.89   73.67  664.83   70.86     673   71.33
#Mann= 5 ,-1 , 0
       0      .1       0  171.44     .07       0  328.57    .035       0
  341.76     .07       0  439.12     .99       0
Bank Sta=171.44,439.12
XS Rating Curve= 0
Exp/Cntr=.3,.1

Type RM Length L Ch R = 1 ,6022.230,52.37,55.07,44.29
BEGIN DESCRIPTION:
D
END DESCRIPTION:
XS GIS Cut Line= 4
     3056930.891     13844408.03     3056675.396    13844174.773
     3056644.874    13844119.567     3056449.268     13843929.95
#Sta/Elev= 30
       0   73.17   52.85   71.49   59.68   71.43   95.53   72.19  176.25   71.07
  191.25   72.11  203.35   72.26  223.06   74.58  225.06   74.65  245.66   74.53
  267.05    72.7  267.56   72.68  288.29   65.06  293.32   64.08  322.68    59.6
  324.65   59.17  346.18    54.3  354.04   50.25  361.04   49.65  370.04   52.15
  379.83   53.96  385.35   55.49  390.83   57.08  409.04   63.05  437.75   71.67
  456.76   73.11  493.81   72.33  520.29   71.52  598.39    72.8  681.47   72.83
#Mann= 5 ,-1 , 0
       0      .1       0  267.05     .07       0  354.04    .035       0
  370.04     .07       0  437.75     .99       0
Bank Sta=267.05,437.75
XS Rating Curve= 0
Exp/Cntr=.5,.3

Type RM Length L Ch R = 1 ,5966.850,7.97,8,7.95
BEGIN DESCRIPTION:
u/s side of Nature Reserve Footbridge, from Klotz
END DESCRIPTION:
XS GIS Cut Line= 4
      3056951.17    13844367.082     3056728.134    13844145.152
     3056689.091    13844099.486     3056469.547    13843889.002
#Sta/Elev= 30
       0   72.71    28.1   72.16   40.83   72.07   104.5   73.47  133.91   73.08
  178.41   71.45  188.52   71.56  208.46   73.52  220.34   73.14  264.03   70.62
  273.38   68.73  319.03   54.75  327.15   52.59  328.69   52.56  338.13   50.25
  341.72   49.04  346.12   49.11  350.11   49.53  354.13   52.15  369.17    61.3
  378.65   63.96  384.62   65.94  400.85   70.02   416.4   70.62  434.52      72
  458.41    71.5  587.45   73.94   612.1   74.16  650.15   74.17  678.86   73.63
#Mann= 6 ,-1 , 0
       0     .99       0    28.1      .1       0  264.03     .07       0
  338.13    .035       0  354.13     .07       0  400.85     .99       0
#XS Ineff= 2 , 0
       0  275.27   70.85  393.41       0   70.85
Permanent Ineff=
       F       F
Bank Sta=264.03,400.85
XS Rating Curve= 0
Exp/Cntr=.5,.3

Type RM Length L Ch R = 3 ,5962.856,,,
BEGIN DESCRIPTION:
Nature Reserve Footbridge
END DESCRIPTION:
Bridge Culvert--1,0,-1,-1, 0
Deck Dist Width WeirC Skew NumUp NumDn MinLoCord MaxHiCord MaxSubmerge Is_Ogee
.01,7.98,2.6,0, 2, 2, 70.85, , .95, 0, 0,0,,
     260     420
   70.85   70.85
   68.15   68.15
     260     420
   70.85   70.85
   68.15   68.15
BR Coef=-1 , 0 , 0 ,, 0 ,,,.8,-1,,0,
WSPro=,,,, 1 ,,,, 0 ,,,, 0 ,,,,-1 ,-1 ,-1 , 0 , 0 , 0 , 0 , 0
BC Design=,, 0 ,, 0 ,,,,,,
BC HTab HWMax=74.17

Type RM Length L Ch R = 1 ,5958.857,22.8,20.5,20.6
BEGIN DESCRIPTION:
d/s side of Nature Reserve Footbridge, from Klotz
END DESCRIPTION:
XS GIS Cut Line= 4
     3056957.224    13844361.869     3056734.188    13844139.939
     3056695.145    13844094.273     3056475.601    13843883.789
#Sta/Elev= 30
       0   72.64      23   72.19   39.81   72.19  109.07   73.69  126.51   73.46
  181.66   71.43  189.12   71.52  213.82   73.94  244.81   72.44  272.57    69.6
  273.97   69.32  281.07   67.14  314.64   58.12  323.76   55.87  337.08   50.25
  340.67   49.04  345.07   49.11  349.06   49.53  371.44   61.85  381.24   64.86
  400.56   69.76     404   70.46  408.83   70.47  424.78   71.08  434.23    71.8
  446.68   71.55  589.18   74.14  618.29   74.41  646.72   74.42  678.86   73.81
#Mann= 6 ,-1 , 0
       0     .99       0   39.81      .1       0  244.81     .07       0
  337.08    .035       0  349.06     .07       0     404     .99       0
#XS Ineff= 2 , 0
       0  277.78   70.85  394.21       0   70.85
Permanent Ineff=
       F       F
Bank Sta=244.81,404
XS Rating Curve= 0
Exp/Cntr=.5,.3

Type RM Length L Ch R = 1 ,5938.748,92.98,83.66,91.59
XS GIS Cut Line= 2
     3056974.462    13844346.604     3056492.839    13843868.524
#Sta/Elev= 29
       0   72.43    7.96   72.27   30.29   72.35   68.04   72.18  122.99    73.8
  190.48   71.39  220.17   74.21  233.13   74.02   238.5   73.14  279.61   69.21
  317.55   63.74  338.94   55.55  339.21   55.54  346.03   50.25  348.03   49.48
  349.62   49.04  351.77   49.14  354.02   49.11  355.79   49.23  358.01   49.53
   360.5   56.51  388.38   65.34  395.72   67.19  403.09   68.69  416.63   72.01
  444.48   72.07  593.41    74.7  635.07    75.1  678.62   74.33
#Mann= 6 ,-1 , 0
       0     .99       0   68.04      .1       0   238.5     .07       0
  346.03    .035       0  358.01     .07       0  416.63     .99       0
Bank Sta=238.5,416.63
XS Rating Curve= 0
Exp/Cntr=.3,.1

Type RM Length L Ch R = 1 ,5853.792,512.06,487.81,366.05
XS GIS Cut Line= 4
     3057115.582    13844295.375     3056815.376      13844084.1
     3056781.171    13844025.304     3056542.834    13843789.521
#Sta/Elev= 30
       0   73.04   24.36   73.22   246.4   72.11  248.02    72.1  270.24    75.7
  312.94   69.02   336.5   68.66   367.1   57.69  373.33   55.07  375.72   50.05
  377.82   49.49  389.19   47.88  393.24    49.1  401.72   49.85  405.54   52.05
  413.18   54.91  435.12   56.95  463.29   61.35  493.83   66.78  497.23   68.01
  518.41   71.03  543.66   72.15  605.79   71.94  634.65   72.53  648.96   71.32
  691.32   71.78  707.24   74.04  720.44   74.57  760.97   73.44  770.38   72.68
#Mann= 6 ,-1 , 0
       0     .99       0   246.4      .1       0   336.5     .07       0
  377.82    .035       0  393.24     .07       0  518.41     .99       0
Bank Sta=336.5,518.41
XS Rating Curve= 0
Exp/Cntr=.3,.1

Type RM Length L Ch R = 1 ,5371.263,69,81.46,84.5
XS GIS Cut Line= 2
     3057476.483    13843851.202     3056470.231     13843432.39
#Sta/Elev= 30
       0   73.35   60.79   73.35  156.56    75.3  176.76   75.07  268.42   72.74
  348.36   72.02   429.1   70.69  437.19   69.66  450.99   67.25  512.96   63.22
  517.11   62.62  552.32   55.75  555.86   54.55  559.76   49.07  566.77   48.31
   572.1   49.06  581.82   55.58  620.86   60.06   625.5   60.17  648.53   65.54
  658.55   67.54  665.05   67.83  674.24   69.92  706.74   71.23  746.55   71.59
  826.79   71.06  876.85   71.43  923.59   71.21 1027.75   73.17 1089.93   72.86
#Mann= 5 ,-1 , 0
       0      .1       0   429.1     .07       0  559.76    .035       0
   572.1     .07       0  674.24     .99       0
Bank Sta=429.1,674.24
XS Rating Curve= 0
Exp/Cntr=.3,.1

Type RM Length L Ch R = 1 ,5285.146,33.97,62.96,83.92
XS GIS Cut Line= 2
     3057441.449    13843773.193     3056435.483    13843304.752
#Sta/Elev= 30
       0   73.93   19.24   74.95   60.63   73.69   77.52   75.04  107.57   73.25
  136.11   75.26   170.4   76.16  210.99   72.59  254.64   73.28  345.72   69.87
  370.91   64.66  398.16   54.68  409.18   53.59  449.45   53.02  461.37   51.62
  482.55   54.37  518.94   54.28  557.06   51.96  559.87   49.18  570.72   46.24
  575.59   48.25  577.04   51.64  596.84   52.95  604.61   56.86  618.84   61.25
  664.55   70.73  739.11   73.46  931.93   73.36  986.01   71.17 1109.69    73.3
#Mann= 5 ,-1 , 0
       0      .1       0  345.72     .07       0  559.87    .035       0
  575.59     .07       0  664.55     .99       0
Bank Sta=345.72,664.55
XS Rating Curve= 0
Exp/Cntr=.3,.1

Type RM Length L Ch R = 1 ,5221.017,176.54,229.02,239.5
XS GIS Cut Line= 2
     3057299.392    13843682.358     3056605.297    13843231.362
#Sta/Elev= 30
       0   76.41   46.04   72.51  147.17   72.56  165.16   72.41  191.27   70.02
  213.74   64.16  227.05   63.07   231.4   61.13   238.1    57.4  244.93   53.86
  256.76   48.52  260.91    46.9  264.41   46.49  271.32   47.63  283.76   52.22
  287.74   53.81  316.49   69.02  326.08   70.12  337.46   67.88  350.67   64.13
  361.35   63.33  372.36   61.19  385.98    60.4  457.02   69.09  594.61   72.09
  601.06   72.09  651.06    73.1  665.12    73.6  812.28   71.32  827.75   70.89
#Mann= 5 ,-1 , 0
       0      .1       0  191.27     .07       0  256.76    .035       0
  271.32     .07       0  316.49     .99       0
#Block Obstruct= 2 , 0
       0                  337.46       0      67
Bank Sta=191.27,326.08
XS Rating Curve= 0
Exp/Cntr=.3,.1

Type RM Length L Ch R = 1 ,4985.114,147.41,417.68,457.86
XS GIS Cut Line= 3
     3057434.115    13843636.302     3057235.016    13843368.262
     3056810.196    13843061.561
#Sta/Elev= 30
       0   72.04   87.57    71.4  123.62   72.94  133.64   73.09     210   69.11
  235.02   63.19   268.1   57.15   274.1   51.85   281.1   48.02   287.6   47.31
  289.97   47.45  292.18   47.16  294.26   47.43   302.1   52.35  324.83   57.83
  340.09   60.45  363.08   60.35  389.86   62.06  410.28   62.95  425.23   66.63
  447.13   68.88  480.15   69.54  544.81   72.57  560.69   72.97  594.05   71.56
  650.65   69.98   697.7    72.5  716.19   72.75  726.76    72.5  857.86   73.59
#Mann= 5 ,-1 , 0
       0      .1       0     210     .07       0   281.1    .035       0
  294.26     .07       0  447.13     .99       0
Bank Sta=210,447.13
XS Rating Curve= 0
Exp/Cntr=.3,.1

Type RM Length L Ch R = 1 ,4569.578,215.71,189.74,43.55
XS GIS Cut Line= 4
     3057436.693    13843535.348     3057382.664    13843154.847
     3057402.101    13843107.649     3057368.841     13842731.39
#Sta/Elev= 30
       0   71.84   12.84      72   45.22   74.13   58.29   73.76   75.59   69.92
   99.49      68  131.18   67.83  171.95   65.03   229.3    69.6  259.57   67.28
  274.73   64.14  292.13    62.6  314.56   59.31     325   59.57  354.39    55.2
  370.27   54.07  405.26   46.98  411.68   45.56  414.39   45.59  418.97   47.11
  435.42   58.16  444.75   58.65  449.78   60.47  460.99   63.06  489.13   68.56
  516.19   69.66  531.02   71.38  610.14   73.61  708.65   70.53  813.09   72.72
#Mann= 5 ,-1 , 0
       0      .1       0   229.3     .07       0  405.26    .035       0
  418.97     .07       0  489.13     .99       0
#Block Obstruct= 2 , 0
       0  194.62      67               0
Bank Sta=229.3,489.13
XS Rating Curve= 0
Exp/Cntr=.3,.1

Type RM Length L Ch R = 1 ,4381.730,157.64,133.76,23.33
BEGIN DESCRIPTION:
C
END DESCRIPTION:
XS GIS Cut Line= 5
     3057694.623    13843594.761     3057573.319     13843228.28
     3057520.137    13843189.367     3057477.333    13843097.272
     3057402.411    13842903.619
#Sta/Elev= 30
       0   73.47   40.63   73.61  180.55   70.84  191.87   72.07  214.96   73.98
  216.63   73.96  252.39   72.92  295.05   69.21  344.26   67.14  366.07   60.36
  372.28   58.33   384.1   56.85  388.99   54.42  408.15   49.51  414.82   48.89
  419.61   48.02  432.56   49.24  444.08   49.54  453.01   50.54  458.52   51.84
  489.76   53.15  509.96    57.4  517.82   59.58  546.05   62.71  589.03   69.21
  623.73   69.58  628.78   70.46  706.39   72.92  728.45   73.13  761.13   71.88
#Mann= 5 ,-1 , 0
       0     .99       0  344.26     .07       0  408.15    .035       0
  432.56     .07       0  589.03     .99       0
Bank Sta=344.26,589.03
XS Rating Curve= 0
Exp/Cntr=.3,.1

Type RM Length L Ch R = 1 ,4260.886,17.52,74.51,135.78
XS GIS Cut Line= 4
     3057901.762    13843508.205     3057599.377    13843100.693
     3057529.217    13843077.816     3057406.412    13842893.617
#Sta/Elev= 30
       0   72.96   43.35   74.17  136.69   70.36  172.44   69.95  202.93   71.18
  272.94   72.46  340.98   71.93  398.99   69.77  438.05   71.39  469.03   67.04
  486.35   59.96  494.31   58.39  499.68   58.66  528.97    57.4     545    54.6
   552.1   52.45  562.95   47.09  565.94   46.67  573.51   46.96  577.45    47.7
  582.51    47.8  588.06   52.84  617.02   59.44  626.37   60.04  637.86   63.39
  663.28   65.16  699.49    66.4  722.23    70.7  768.95   72.25  802.63   71.48
#Mann= 5 ,-1 , 0
       0     .99       0  438.05     .07       0  562.95    .035       0
  582.51     .07       0  722.23     .99       0
Bank Sta=438.05,722.23
XS Rating Curve= 0
Exp/Cntr=.3,.1

Type RM Length L Ch R = 1 ,4203.385,126.91,200.19,160.74
XS GIS Cut Line= 5
     3057905.281    13843504.689     3057604.321    13843052.383
     3057579.228    13842998.014     3057527.213    13842787.247
     3057469.496    13842601.352
#Sta/Elev= 30
       0    73.1   46.72   74.09  135.55   70.53   191.7   69.75  273.94   72.74
  359.74   71.91  435.21    69.3  449.36   69.84  459.64   68.39  494.38   57.61
  527.75   56.01  534.47   53.96   544.6   48.19  547.23   47.38  552.19   46.59
  562.07   47.63  568.76   51.51  575.23    56.7  580.74   58.82  591.65   60.95
  621.08   60.34  638.16   60.86  652.21   60.04  690.79   63.03  710.72   66.11
  725.68   70.74   799.2   72.11  873.46   72.05  934.91   70.47  1014.9   72.06
#Mann= 5 ,-1 , 0
       0     .99       0  449.36     .07       0  547.23    .035       0
  562.07     .07       0  725.68     .99       0
Bank Sta=449.36,725.68
XS Rating Curve= 0
Exp/Cntr=.3,.1

Type RM Length L Ch R = 1 ,3991.037,199.29,189.28,165.35
XS GIS Cut Line= 4
      3058249.56    13844233.656     3057754.881    13842920.643
     3057727.696    13842874.639     3057544.498    13842561.336
#Sta/Elev= 30
       0    74.1    54.6   71.72  209.65   76.03  326.71   75.26  389.27   71.24
  476.18   74.91  639.21   72.62  709.48   70.41  794.84   73.61  921.21   73.19
 1130.81   68.88 1198.18   69.87 1258.76   68.72  1324.8   68.84 1353.47    65.1
 1388.34   59.14 1399.84   52.85 1402.84   47.95 1408.78   45.27 1411.75   45.25
 1416.97   46.67 1430.16   55.35 1449.83    57.9 1466.55   58.36 1502.66   62.04
 1557.05   69.59 1635.78   72.14 1642.08   71.42 1727.74   72.83 1819.48   71.72
#Mann= 5 ,-1 , 0
       0     .99       0  1324.8     .07       0 1402.84    .035       0
 1416.97     .07       0 1557.05     .99       0
Bank Sta=1324.8,1557.05
XS Rating Curve= 0
Exp/Cntr=.3,.1

Type RM Length L Ch R = 1 ,3804.938,189.51,116.15,111.09
XS GIS Cut Line= 4
     3058118.609    13843360.494     3057903.071    13842827.419
     3057879.635    13842772.502     3057513.235    13842304.415
#Sta/Elev= 30
       0   73.93   19.27   74.08   90.38   69.69  160.86   71.11  283.29   70.57
  362.89   68.36  504.38   69.31  558.76   67.14  570.93   52.68  581.02   46.48
  583.17   46.06  588.32   46.08  593.18   45.23  600.68   46.52  603.19   51.73
  610.83   55.38  618.26   57.12  623.67   55.42  635.37   57.94  672.64   62.09
  679.88   62.77  696.52      62  732.02   66.42  805.85   68.11  882.18   70.84
 1004.62   71.14 1034.57   70.47  1088.9   71.92 1179.22   70.69 1229.15   72.08
#Mann= 5 ,-1 , 0
       0     .99       0  504.38     .07       0  583.17    .035       0
  600.68     .07       0  882.18     .99       0
Bank Sta=504.38,732.02
XS Rating Curve= 0
Exp/Cntr=.3,.1

Type RM Length L Ch R = 1 ,3678.735,224.85,224.22,132.16
XS GIS Cut Line= 4
     3058570.324    13843561.518     3057970.264    13842715.715
     3057951.445     13842667.62     3057571.149    13842242.383
#Sta/Elev= 30
       0   71.46   125.3   74.54  141.57   72.51  237.58   73.37  329.05   69.42
  399.14   72.37  452.99   72.82  594.97   71.82  654.01   68.84  713.39   67.95
  760.07   69.84  773.23   69.88  793.25   67.78  876.11   70.13  974.71   68.51
 1047.85   55.17  1061.8   51.76 1066.95    45.9  1070.1   45.46 1077.08   45.21
 1084.29   45.76 1114.65   56.04 1144.56   60.97 1166.67   63.25 1201.12   69.54
 1225.72   70.41 1398.22   70.16 1490.42   73.47 1574.64   73.75 1659.17   71.78
#Mann= 5 ,-1 , 0
       0     .99       0  974.71     .07       0  1070.1    .035       0
 1084.29     .07       0 1201.12     .99       0
Bank Sta=974.71,1201.12
XS Rating Curve= 0
Exp/Cntr=.3,.1

Type RM Length L Ch R = 1 ,3470.650,369.82,492.03,496.73
BEGIN DESCRIPTION:
Beltway 8 area blocked
END DESCRIPTION:
XS GIS Cut Line= 4
     3058757.785    13843429.181     3058104.095    13842540.062
     3058045.544     13842517.06     3057619.967    13842222.207
#Sta/Elev= 30
       0   67.99     8.8   72.51  152.22   70.72  236.93   70.83  272.18   73.83
  318.88   71.83   452.9   69.46  487.54   69.76  507.99   68.63  621.08   71.38
  753.16   70.86  821.56   68.02  995.31   69.41 1040.39   66.88  1072.1    56.9
 1082.69   44.21 1091.85   42.82 1094.34   43.45 1114.38   55.21 1125.69   60.35
 1134.69   56.35 1145.69   54.95 1163.69   59.55 1178.69   60.55 1201.69   59.85
 1275.44   70.33 1288.87   70.91 1426.55    69.6 1476.31   72.23 1684.21   73.93
#Mann= 5 ,-1 , 0
       0     .99       0  995.31     .07       0 1082.69    .035       0
 1094.34     .07       0 1275.44     .99       0
#Block Obstruct= 2 , 0
       0     8.8   72.51               0
Bank Sta=995.31,1275.44
XS Rating Curve= 0
Exp/Cntr=.3,.1

Type RM Length L Ch R = 1 ,2972.127,515.87,614.27,574.29
BEGIN DESCRIPTION:
B
END DESCRIPTION:
XS GIS Cut Line= 4
     3058791.512    13842933.529     3058290.204    13842126.023
     3058245.312    13842065.543      3057503.34    13841497.864
#Sta/Elev= 30
       0   70.66   28.25   71.45  209.74   70.36   306.5   67.57  410.52   71.39
  661.72    67.8  737.79    71.5  824.72   69.49  857.93   67.24  884.81   65.82
  918.62   58.22  927.59   57.98  954.86   52.33  955.29   52.19  959.15   42.89
  966.17   40.85   982.5   42.58  983.15   45.35  991.87   52.05 1010.37   54.95
 1036.69    68.1 1115.21   71.22 1207.28    71.4 1392.52   69.09 1449.36   71.56
 1510.76   69.17 1693.91   68.43 1820.49   71.98 1937.22   67.26 1960.01   68.03
#Mann= 5 ,-1 , 0
       0     .99       0  857.93     .07       0  959.15    .035       0
   982.5     .07       0 1036.69     .99       0
Bank Sta=857.93,1036.69
XS Rating Curve= 0
Exp/Cntr=.3,.1

Type RM Length L Ch R = 1 ,2360.236,370.38,330.55,237.58
BEGIN DESCRIPTION:
Beltway 8 area blocked
END DESCRIPTION:
XS GIS Cut Line= 4
     3059217.564    13842755.121     3058873.622     13842063.29
     3058838.698    13842004.545     3058393.867    13841402.325
#Sta/Elev= 30
       0   68.28   68.72   69.28   83.94   67.38   95.28   54.21  106.61   49.29
  130.12   45.51  299.36   49.24  319.73    66.2  330.54   69.37  418.85   66.21
   583.9   68.53  603.87   65.58  639.14   64.25  684.86   57.19  723.84   48.52
   737.9   51.91  760.76   49.82  768.04   47.41   837.6   49.27  845.74   42.35
  853.21   41.58  859.68   42.24  874.56   51.02  908.01   53.52  950.78   65.95
  982.96   67.68 1146.26   67.12 1250.17   69.78 1513.62   72.03 1589.65   66.45
#Mann= 5 ,-1 , 0
       0     .99       0   583.9     .07       0  845.74    .035       0
  859.68     .07       0  982.96     .99       0
#Block Obstruct= 2 , 0
       0  330.54   69.37               0
Bank Sta=583.9,982.96
XS Rating Curve= 0
Exp/Cntr=.3,.1

Type RM Length L Ch R = 1 ,2022.700,236.5,157.54,137.69
XS GIS Cut Line= 4
     3059275.507    13842058.003     3059043.002    13841762.171
     3058988.205    13841718.563     3058490.095    13841376.491
#Sta/Elev= 30
       0   67.03  113.59   65.27  124.57   65.59  219.68   70.51  230.51   70.17
  296.41   70.72  334.89   66.91  359.41   60.08  373.47   55.68  392.77   51.34
  405.48   50.02  418.74   42.75  420.74   41.25  424.49   40.52   427.3   40.68
  441.74   49.55  449.74   52.15  450.92   53.38  483.67   62.26  488.78   63.87
   541.9   70.48  558.81   70.44  586.16   68.96  635.49   68.96  714.94   70.12
  736.35   70.78  814.85   66.29  912.15   70.63 1039.27   72.68 1050.55   72.22
#Mann= 5 ,-1 , 0
       0     .99       0  296.41     .07       0  418.74    .035       0
   427.3     .07       0   541.9     .99       0
Bank Sta=296.41,541.9
XS Rating Curve= 0
Exp/Cntr=.3,.1

Type RM Length L Ch R = 1 ,1866.190,97.42,210.95,135.96
BEGIN DESCRIPTION:
adjusted for skewness
END DESCRIPTION:
XS GIS Cut Line= 5
     3059337.847    13841766.353     3059310.366    13841725.045
     3059145.466    13841645.069     3059080.641    13841592.791
     3058449.764    13841233.504
#Sta/Elev= 30
       0   69.56   36.91   70.37   61.58   69.18  121.81   70.16  155.12   69.69
  188.09   67.38  233.18   53.01  246.65   50.29  266.07    51.9  328.97   51.26
  353.82   56.58  366.41   56.85  369.93   54.79  391.93   53.23   396.4   47.06
  403.43   41.22  408.56   39.88  417.32   41.57  423.14   51.83  448.88   55.46
  473.95   62.66  499.57   65.55  511.38   68.53  668.27   70.89  745.05   66.03
  810.32   70.93  924.17   72.46  955.51   70.76 1002.96   54.41 1042.17   54.06
#Mann= 5 ,-1 , 0
       0     .99       0  155.12     .07       0  403.43    .035       0
  417.32     .07       0  511.38     .99       0
#Block Obstruct= 2 , 0
       0                  955.51       0   70.76
Bank Sta=155.12,511.38
XS Rating Curve= 0
Exp/Cntr=.3,.1

Type RM Length L Ch R = 1 ,1681.007,25.38,210.59,211.92
XS GIS Cut Line= 4
     3059352.479    13841758.898     3059216.563    13841444.323
      3059128.31     13841432.06      3058553.14    13841197.505
#Sta/Elev= 30
       0   70.37   28.97   69.31   49.71   70.32   87.65   68.07  127.08   68.07
  188.33   69.53   330.4   67.19  377.89   60.74  391.19   52.95  406.93   41.33
     412   41.06  416.09   39.46  422.19   39.28  428.07   40.43  440.19   49.55
  473.93   60.19  519.96   65.38  556.03   67.85  625.02   68.45  645.72   69.32
  714.07   68.73  786.01    69.4  842.66    71.5  893.58   66.32  916.39   65.71
  946.61   70.59 1003.25   71.07 1011.94   69.56 1049.63   69.79 1052.94    67.3
#Mann= 5 ,-1 , 0
       0     .99       0   330.4     .07       0     412    .035       0
  428.07     .07       0  556.03     .99       0
Bank Sta=330.4,556.03
XS Rating Curve= 0
Exp/Cntr=.3,.1

Type RM Length L Ch R = 1 ,1481.135,47.37,256.27,497.52
BEGIN DESCRIPTION:
Other ditch system to the Buffalo Bayou blocked
END DESCRIPTION:
XS GIS Cut Line= 5
     3059388.034     13841931.55     3059378.249    13841825.314
     3059212.381     13841249.85     3059164.286    13841214.301
     3058607.526    13841002.562
#Sta/Elev= 30
       0   70.45   44.95   71.12  155.91   69.58  170.75   70.28  219.54   67.44
  309.82   68.99  441.18   68.14  464.46   67.32  506.13   60.27  535.41   57.57
  540.36   56.34  583.74   57.38  642.15   54.37  651.15   51.85  661.15   41.75
  672.26   40.78  681.15   42.05  701.24   52.83   734.5   60.21  751.75   67.08
  777.47   69.86  831.89   69.48  874.56    67.4  912.91   69.93  987.92   69.74
 1024.22   68.21 1136.41   68.45 1224.94   59.77 1264.64   52.04 1361.05   50.79
#Mann= 5 ,-1 , 0
       0     .99       0  441.18     .07       0  661.15    .035       0
  681.15     .07       0  777.47     .99       0
#Block Obstruct= 2 , 0
       0                 1136.41       0   68.45
Bank Sta=441.18,777.47
XS Rating Curve= 0
Exp/Cntr=.3,.1

Type RM Length L Ch R = 1 ,1246.119,49.59,74.8,51.21
BEGIN DESCRIPTION:
A
END DESCRIPTION:
XS GIS Cut Line= 4
     3059403.092    13841939.355     3059342.292    13841398.255
      3059420.91    13841290.879     3059488.026    13840734.969
#Sta/Elev= 30
       0   69.57  112.43   71.09  293.56   69.64  336.79   65.89  407.96   67.32
  500.91   65.48  518.81   64.24  534.47   58.56  545.56   55.96  560.27   49.46
  564.58   48.52  573.68   48.45  579.02   40.81  581.84   39.89  590.41   39.81
  593.25    40.7  599.98   41.24  608.92   47.75  647.92   65.42  660.86   66.53
  665.79   67.76  838.59   68.17  885.84   69.75  915.24      72 1015.83   70.93
 1054.84   73.28 1114.85   70.72  1128.6   69.35 1206.47   66.84 1237.53   68.91
#Mann= 6 ,-1 , 0
       0     .99       0  407.96     .07       0  579.02    .035       0
  599.98     .07       0  660.86     .05       0  838.59     .99       0
Bank Sta=500.91,660.86
XS Rating Curve= 0
Exp/Cntr=.5,.3

Type RM Length L Ch R = 1 ,1170.684,12.95,14.02,13.53
BEGIN DESCRIPTION:
u/s face of Wastewater Treatment Bridge
END DESCRIPTION:
XS GIS Cut Line= 5
     3059419.852    13842010.273      3059415.09    13841449.786
     3059473.197    13841311.274     3059483.915    13841289.697
     3059510.353    13840765.467
#Sta/Elev= 30
       0   62.94   33.21      69  182.65   71.01  336.76   69.07  366.12   70.35
  408.28   69.55  443.63   66.82  486.05   64.79  550.21   63.87  557.36  64.705
  568.22   63.35  569.19   61.58  576.44   59.65  582.41   56.27  590.79   53.53
  595.47   48.86  599.82   48.54   620.4   40.75  630.08   40.12  637.26   40.75
  652.92   47.73  675.49   55.14  685.32   63.35  715.22   66.05  930.81   68.52
  993.67   72.55 1032.35   72.08 1049.68   73.04 1169.47   70.56  1259.7   67.44
#Mann= 6 ,-1 , 0
       0     .99       0  443.63     .07       0   620.4    .035       0
  637.26     .07       0  715.22     .05       0  930.81     .99       0
#XS Ineff= 2 , 0
       0  560.51   63.94  685.32       0   66.25
Permanent Ineff=
       F       F
#Block Obstruct= 2 , 0
       0   33.21      69               0
Bank Sta=557.36,715.22
XS Rating Curve= 0
Exp/Cntr=.5,.3
